--- ZEBSCK.prj (project) ---

Proj Title=ZEBSCK
Current Plan=p01
Default Exp/Contr=0,0
English Units
Geom File=g01
Flow File=f01
Plan File=p01
BEGIN DESCRIPTION:
END DESCRIPTION:
DSS Export Rating Curves= 0
DSS Export Rating Curve Sorted= 0
DSS Export Volume Flow Curves= 0
DXF OffsetX= 0
DXF OffsetY= 0
DXF ScaleX= 0
DXF ScaleY= 0

--- ZEBSCK.p01 (plan) ---

Plan Title=Floodplain
Program Version=4.00
Geom File=g01
Flow File=f01
K Sum by GR=0
Std Step Tol=0.01
Critical Tol=0.01
Num of Std Step Trials=20
Max Error Tol=0.3
Flow Tol Ratio=0.001
Split Flow NTrial=30
Split Flow Tol=0.02
Split Flow Ratio=0.02
Log Output Level=0
Friction Slope Method=1
Unsteady Friction Slope Method=2
Unsteady Bridges Friction Slope Method=1
Global Log Level=0
CheckData=False
Run HTab=0
Run UNet=0
Run PostProcess=0
UNET Theta=0
UNET Theta Warmup=0
UNET ZTol=0
UNET ZSATol=0
UNET MxIter=0
UNET MaxInSteps=0
UNET DtIC=0
UNET DtMin=0
UNET MaxCRTS=0
UNET WFStab=0
UNET SFStab=0
UNET WFX=0
UNET SFX=0
UNET DSS MLevel=0
UNET DZMax Abort=0
UNET Convert EG Bridges=0
UNET Use Existing IB Tables=0
UNET Froude Limit=0
UNET Froude Power=0
Write IC File=0
Echo Input=False
Echo Output=False
Write Detailed=0

--- ZEBSCK.f01 (steady flow) ---

Flow Title=NFF Regression Equation
Program Version=4.10
Number of Profiles= 1
Profile Names=P100yr
River Rch & RM=ZEBSCK,Main            ,16191.8
553.6898
River Rch & RM=ZEBSCK,Main            ,12904.6
 609.114
River Rch & RM=ZEBSCK,Main            ,12611.9
787.3117
River Rch & RM=ZEBSCK,Main            ,10992
828.7164
River Rch & RM=ZEBSCK,Main            ,8788.6
894.1901
River Rch & RM=ZEBSCK,Main            ,2981.1
971.7225
River Rch & RM=ZEBSCK,Main            ,2530.5
1210.251
River Rch & RM=ZEBSCK,Main            ,475.1
1235.221
River Rch & RM=ZEBSCK,Main            ,268.7
1236.785
Boundary for River Rch & Prof#=ZEBSCK,Main            , 1
Up Type= 0
Dn Type= 3
Dn Slope=0.015
DSS Import GetInterval= 0
DSS Import GetPeak= 0
DSS Import FillOption= 0

--- ZEBSCK.g01 (geometry) ---

Geom Title=USGS 10m DEM
Program Version=4.10

River Reach=ZEBSCK          ,Main
Reach XY= 30
     1828937.937      182093.513     1829084.598      181786.209
     1828932.086      181132.396     1828976.961      180915.471
     1829594.489      180211.221     1830305.021      179790.249
     1830213.785      179331.079     1830317.644      179200.979
     1830317.366      178784.415     1830193.072      178372.751
      1830264.75      178021.625     1830609.998      177662.752
     1830575.125      176873.654     1830864.889      176399.435
     1830858.748      175901.092     1831145.248      175475.655
     1831083.447      175146.798     1831207.132      174991.091
     1831139.002       174524.69     1831215.585      174361.825
     1831036.377      174090.765     1831569.501      173449.125
     1831583.501      172801.953     1831866.375      172522.968
     1831701.251      172088.892     1831796.825      171719.784
     1830961.375      170453.015     1831057.749       169522.92
       1831225.5      169021.547     1831245.581      168339.917

Type RM Length L Ch R = 1 ,16191.8 ,314.2,304.4,294.1
XS GIS Cut Line= 3
     1829098.793      182146.215     1829039.268        182146.3
     1828780.963      181979.807
#Sta/Elev= 22
       0 1945.09      17 1939.64    25.5 1937.11      51 1930.06    59.5 1928.04
    69.1 1926.39    78.7 1925.56    88.3 1925.14   117.2 1924.04     146 1923.09
   155.6 1922.79   165.2 1922.64   174.8 1922.71   184.4 1923.03     194 1923.45
   232.4 1924.84   299.6 1927.61  328.071928.491     338 1928.54   347.6 1928.06
   357.2 1927.07   366.8 1926.33
#Mann= 4 ,-1 , 0
       0     .12       0     146    .045       0   184.4     .12       0
  328.07    .016       0
Bank Sta=146,184.4
XS Rating Curve= 0 ,0
Exp/Cntr=0.3,0.1

Type RM Length L Ch R = 1 ,15887.4 ,221.9,203.2,183.9
XS GIS Cut Line= 2
     1829140.303      181901.214     1828862.371      181794.796
#Sta/Elev= 24
       0 1944.52     9.6 1942.01    19.2 1938.49   28.311934.296    38.4  1930.2
      48 1927.78    57.6 1926.58    67.2 1925.85   105.6 1923.28   115.2 1922.46
   124.8 1921.52   129.6 1921.18   134.4 1920.83     144 1920.74   153.6 1920.87
   163.2  1921.1  168.411921.219   182.4 1921.55     192  1921.9   216.51923.076
     240 1923.92   259.2 1924.46  281.231925.331   297.6 1926.23
#Mann= 7 ,-1 , 0
       0    .016       0   28.31     .12       0   129.6    .045       0
   163.2     .12       0  168.41    .016       0   216.5     .06       0
  281.23     .12       0
Bank Sta=129.6,163.2
XS Rating Curve= 0 ,0
Exp/Cntr=0.3,0.1

Type RM Length L Ch R = 1 ,15684.2 ,82.5,83.7,84.3
XS GIS Cut Line= 4
     1829171.169      181680.703     1829160.146      181676.362
     1828967.004      181698.498     1828896.621      181674.959
#Sta/Elev= 25
       0 1933.13    5.45 1931.44    11.8 1929.72    21.6 1928.12    31.3 1927.03
      41  1925.6    50.7 1923.94   53.941923.309    60.4 1922.05    79.9 1917.57
      83 1917.24    89.6 1916.55    99.3 1916.75   118.8 1916.62   128.5  1916.9
  132.721917.118   167.4 1919.09   177.1 1919.55   186.8  1919.9   234.1    1921
   243.4 1921.34   252.6  1922.1   261.9 1923.72   271.2 1926.39   280.5 1929.65
#Mann= 6 ,-1 , 0
       0     .12       0    5.45    .016       0   53.94     .12       0
      83    .045       0   118.8    .016       0  132.72     .12       0
Bank Sta=83,118.8
XS Rating Curve= 0 ,0
Exp/Cntr=0.3,0.1

Type RM Length L Ch R = 1 ,15600.4 ,109.5,112.9,116.8
XS GIS Cut Line= 4
      1829178.65      181599.909     1829164.486      181594.331
     1828971.344      181616.466     1828914.415      181597.427
#Sta/Elev= 28
       0 1929.54    4.72 1928.41     7.6 1927.72    15.2  1926.4    24.9 1925.38
   32.891924.703    44.4 1923.63    73.5 1920.67    83.3 1919.56   102.7 1916.93
   110.7 1916.26   112.4 1916.12   122.2 1915.89   131.9 1915.95   141.6  1916.2
   151.3 1916.62     161 1917.14   170.8 1917.76   180.5 1918.56   190.2 1919.56
   199.9 1920.84   209.6 1922.58   218.2 1925.26   226.8 1928.41   235.4 1931.68
   243.9 1934.77   252.5 1937.63   269.7 1943.07
#Mann= 5 ,-1 , 0
       0     .12       0    4.72    .016       0   32.89     .06       0
   110.7    .045       0   141.6     .12       0
Bank Sta=110.7,141.6
XS Rating Curve= 0 ,0
Exp/Cntr=0.3,0.1

Type RM Length L Ch R = 1 ,15487.5 ,199.8,190.2,181.2
XS GIS Cut Line= 2
     1829174.027       181495.59     1828917.525       181495.59
#Sta/Elev= 18
       0 1926.23   20.211924.873      76 1919.98    85.5 1919.02      95 1917.75
   104.5 1916.05     114 1914.71   123.5 1914.98     133  1916.5   142.5 1918.09
     152 1919.31     171 1921.29   180.5 1922.58     190  1924.2   199.5 1926.62
     209 1930.08   237.5 1941.94   256.5 1949.57
#Mann= 4 ,-1 , 0
       0    .016       0   20.21     .12       0   104.5    .045       0
     133     .12       0
Bank Sta=104.5,133
XS Rating Curve= 0 ,0
Exp/Cntr=0.3,0.1

Type RM Length L Ch R = 1 ,15297.3 ,273.1,284.4,294.9
XS GIS Cut Line= 2
      1829154.53      181276.326     1828876.357      181362.145
#Sta/Elev= 23
       0 1926.79     9.7 1926.06    29.1 1924.36    48.5 1922.93    58.2 1922.08
    67.9 1921.03    77.6 1919.77    87.3 1918.32      97 1916.74   116.4 1913.16
   126.2 1911.56   135.8 1910.41   145.6 1909.82   155.3 1910.01     165 1911.01
   194.1 1915.19   203.8 1917.19   213.5  1920.1   242.6 1930.12   252.3 1933.37
     262 1936.51   271.7 1939.54   291.1 1945.44
#Mann= 3 ,-1 , 0
       0     .12       0   135.8    .045       0     165     .12       0
Bank Sta=135.8,165
XS Rating Curve= 0 ,0
Exp/Cntr=0.3,0.1

Type RM Length L Ch R = 1 ,15012.9 ,145,165.7,186.3
XS GIS Cut Line= 3
     1829164.898      181107.903     1829011.924      181062.967
     1828846.556      181056.117
#Sta/Elev= 24
       0 1918.12     9.4 1916.45    18.8 1914.93    28.1 1913.88    37.5  1913.4
    46.9 1913.18    56.3 1912.85      75 1911.61    84.4  1911.1    93.8 1910.83
   103.2 1910.79   150.1  1911.2   198.4 1911.84   208.1 1911.37   217.8 1909.39
   227.6 1907.06   237.3  1907.2   247.1 1910.33   256.8 1914.93   266.5 1919.37
   295.7 1931.83   305.5 1935.93   315.2 1939.85     325 1943.52
#Mann= 3 ,-1 , 0
       0     .12       0   217.8    .045       0   247.1     .12       0
#XS Ineff= 2 , 0
          197.85 1933.15
Permanent Ineff=
       F       F
Bank Sta=217.8,247.1
XS Rating Curve= 0 ,0
Exp/Cntr=0.3,0.1

Type RM Length L Ch R = 1 ,14847.2 ,187.2,192.3,185.5
XS GIS Cut Line= 2
     1829176.422       181031.18     1828906.332      180850.022
#Sta/Elev= 23
       0 1915.28     9.6 1914.21    19.1  1913.5    47.8 1911.77    76.5 1910.31
    86.1 1909.98    95.6 1909.85   124.4 1909.69   172.2 1909.16   191.3 1908.85
   200.9 1908.34   210.4 1907.49     220 1906.44   229.6 1905.99   239.1 1907.76
   248.7 1911.89   258.3 1917.16   267.8  1922.1   277.4  1926.3     287 1930.19
   296.5 1933.59   306.1 1936.84   325.2 1942.87
#Mann= 3 ,-1 , 0
       0     .12       0   210.4    .045       0   239.1     .12       0
Bank Sta=210.4,239.1
XS Rating Curve= 0 ,0
Exp/Cntr=0.3,0.1

Type RM Length L Ch R = 1 ,14654.9 ,199,200.3,213.4
XS GIS Cut Line= 3
     1829291.465       180918.47     1829095.556      180744.876
     1828960.162      180740.219
#Sta/Elev= 30
       0 1922.64     9.7 1919.85    19.4  1917.5    29.1 1915.39    38.8  1913.7
    48.5 1912.22    67.9 1909.69    77.6 1908.94    87.2 1908.58      97 1908.54
   116.3 1908.75     126 1908.69   135.7 1908.41   145.4  1907.8   193.9 1903.85
   203.6 1903.36   213.3 1903.45   232.7 1904.05   242.4 1904.87   252.1 1907.59
   261.8 1912.68   271.4 1916.31   281.1 1918.96   319.8 1926.53   329.5 1928.86
   348.8  1934.2   358.5 1937.05   368.2 1940.31   387.6 1947.31   397.2 1950.24
#Mann= 3 ,-1 , 0
       0     .12       0   193.9    .045       0   242.4     .12       0
Bank Sta=193.9,242.4
XS Rating Curve= 0 ,0
Exp/Cntr=0.3,0.1

Type RM Length L Ch R = 1 ,14454.6 ,153.5,155,156.5
XS GIS Cut Line= 3
     1829422.617      180778.061     1829273.964      180637.694
     1829127.982       180499.36
#Sta/Elev= 30
       0 1933.72     9.7 1928.91    19.5 1923.54    29.2 1918.69    38.9 1915.16
    48.7 1913.07    87.6    1907   107.1 1904.08   116.8 1902.93   126.6 1902.54
     146  1902.5   155.8 1902.57   194.7 1903.15   204.4 1903.14     214  1902.7
   223.6 1902.16   233.2 1901.99   242.8 1902.03   252.3 1902.23   261.9 1902.84
   281.1 1904.47   290.6 1905.38   300.2 1906.66   309.8 1908.26   338.5 1913.43
   348.1  1915.6   357.7 1918.42   376.8  1924.5     396 1930.18   405.6 1933.29
#Mann= 3 ,-1 , 0
       0     .12       0     214    .045       0   261.9     .12       0
Bank Sta=214,261.9
XS Rating Curve= 0 ,0
Exp/Cntr=0.3,0.1

Type RM Length L Ch R = 1 ,14299.6 ,205.4,206.7,204.3
XS GIS Cut Line= 3
     1829517.812      180672.776     1829307.933      180455.659
     1829278.663      180326.305
#Sta/Elev= 30
       0 1936.58     9.7  1933.4    19.5 1929.56      39 1921.27    48.7 1917.36
    58.4 1914.03    68.2 1911.68    77.9 1909.96   126.6 1902.94   136.4 1902.21
   146.1 1902.06   175.3 1902.13   185.1 1901.95   204.6 1901.46     224 1902.18
   243.5 1903.24     263 1903.85   292.2 1905.38   311.4  1906.8   330.4 1908.72
   339.9 1909.17   349.3 1910.14   358.8 1914.94   368.3  1920.5   377.8 1925.02
   387.2 1928.23   406.2 1933.11   415.6 1935.86   425.1 1938.99   434.6 1942.31
#Mann= 3 ,-1 , 0
       0     .12       0   185.1    .045       0     224     .12       0
Bank Sta=185.1,224
XS Rating Curve= 0 ,0
Exp/Cntr=0.3,0.1

Type RM Length L Ch R = 1 ,14093   ,185.9,171,155.6
XS GIS Cut Line= 3
     1829640.423      180531.433     1829480.385      180373.834
     1829366.614      180259.065
#Sta/Elev= 30
       0 1925.72     9.8 1923.95    19.5 1922.35    48.8 1917.98   61.081915.882
    68.4 1914.44    87.9 1910.14   117.2 1903.86     127 1901.61   136.7 1899.99
   146.5 1899.44     166 1899.47   185.6 1899.78   195.3  1899.8   205.1 1899.49
   217.1 1898.79   234.1 1898.13   243.6 1898.14   253.1 1898.76   262.6 1899.79
   272.1 1901.41   281.6 1904.55   291.2 1907.89   300.7 1911.72   310.2 1916.03
   329.2 1924.95   357.7 1939.06   367.2 1943.62   376.7 1947.52   386.2 1950.58
#Mann= 4 ,-1 , 0
       0     .06       0   61.08     .12       0   217.1    .045       0
   253.1     .12       0
Bank Sta=217.1,253.1
XS Rating Curve= 0 ,0
Exp/Cntr=0.3,0.1

Type RM Length L Ch R = 1 ,13922   ,133.5,157,178.8
XS GIS Cut Line= 4
      1829754.15      180396.307     1829653.851      180283.019
     1829549.684      180246.561     1829473.297      180175.711
#Sta/Elev= 25
       0 1922.45    18.9 1918.33    56.7  1910.3    66.2  1908.4    75.6 1906.73
    85.1  1905.8    94.6 1905.14     104 1904.62   118.21903.975   132.4 1903.43
   169.7  1902.5   188.1  1901.9   197.3  1901.4   206.5 1900.68   215.7 1899.89
   224.9 1899.52   234.1 1900.09   243.3 1901.75   261.7  1905.8   271.1 1908.09
     309 1917.99     328 1922.64   337.4 1924.87   356.4  1929.1   365.9 1930.92
#Mann= 4 ,-1 , 0
       0     .06       0   118.2     .12       0   206.5    .045       0
   243.3     .12       0
Bank Sta=206.5,243.3
XS Rating Curve= 0 ,0
Exp/Cntr=0.3,0.1

Type RM Length L Ch R = 1 ,13765   ,157.7,154.8,154.1
XS GIS Cut Line= 2
     1829814.081      180329.091      1829603.61      180042.377
#Sta/Elev= 27
       0 1922.06     9.6 1920.05    28.8 1916.38    76.9 1907.75    86.5 1906.17
   88.581905.958    96.1 1905.19   105.7 1904.51   115.4 1903.94   134.6  1902.9
   182.6 1900.48   192.3 1899.82   201.9 1898.88   211.3 1898.12   221.1 1897.91
   230.7  1898.9   240.3  1901.1   249.9 1903.91   259.6 1907.29   269.2 1910.96
   278.8 1915.39   288.4 1919.68     298 1923.84   307.6 1927.36   326.8 1933.51
   346.1 1940.15   355.7 1943.26
#Mann= 4 ,-1 , 0
       0     .06       0   88.58     .12       0   201.9    .045       0
   230.7     .12       0
Bank Sta=201.9,230.7
XS Rating Curve= 0 ,0
Exp/Cntr=0.3,0.1

Type RM Length L Ch R = 1 ,13610.1 ,158,170.2,173.5
XS GIS Cut Line= 2
      1829928.15      180266.194     1829713.461       179944.16
#Sta/Elev= 26
       0 1926.83    19.4 1921.38      29  1918.6    38.7  1916.2    48.4 1914.31
    67.7 1911.08    96.8 1906.43   106.4 1904.93   125.8 1902.13   145.1 1899.12
   154.8 1897.91   164.5 1897.39   174.2 1897.36   212.9 1897.36   222.6  1897.4
   232.2 1897.69   241.9 1898.46   251.6 1899.84   261.2  1902.2   280.6  1908.1
     300 1912.93   309.6  1915.5   319.3 1918.23     358 1929.53   367.7 1932.43
     387 1938.42
#Mann= 3 ,-1 , 0
       0     .12       0   174.2    .045       0   212.9     .12       0
Bank Sta=174.2,212.9
XS Rating Curve= 0 ,0
Exp/Cntr=0.3,0.1

Type RM Length L Ch R = 1 ,13440   ,233.1,238.4,256.7
XS GIS Cut Line= 2
     1830064.753      180211.535     1829854.774      179837.279
#Sta/Elev= 26
       0 1933.94     9.8 1931.04    19.5 1928.49    29.3 1926.24    68.3 1917.85
   82.591914.636    97.5 1911.16   136.5 1901.53   146.3 1899.34     156 1897.91
   165.8 1897.43   175.6 1897.36   204.8 1897.36   282.8 1897.35   292.6 1897.36
   302.4  1898.2   312.1  1899.8   321.8 1901.86   331.6  1904.2   341.4 1906.92
   351.1 1910.03   370.6 1916.52   390.1  1922.6   399.9 1925.78   409.6 1929.23
   429.1 1936.54
#Mann= 4 ,-1 , 0
       0     .06       0   82.59     .12       0   165.8    .045       0
   204.8     .12       0
Bank Sta=165.8,204.8
XS Rating Curve= 0 ,0
Exp/Cntr=0.3,0.1

Type RM Length L Ch R = 1 ,13201.5 ,325.3,296.9,242.3
XS GIS Cut Line= 4
     1830213.728      180122.899      1830203.33       179990.05
     1830073.999      179867.971     1829946.391      179754.418
#Sta/Elev= 30
       0  1918.9     9.5 1917.26    57.1  1910.7    66.6 1909.08    95.2 1903.08
   104.7 1901.48   114.2 1900.37   123.7 1899.66   180.1 1897.21   189.4 1896.42
   206.71894.621   217.5 1894.06   226.9 1893.97   236.2 1894.24   245.6 1895.03
   254.9 1896.06   264.3 1896.55   273.7 1896.35     283 1896.65   292.4 1898.25
   301.7 1899.03   311.1 1899.45   358.6 1900.59     387 1901.68   396.5 1902.25
     406  1903.9   415.5 1906.57     444 1915.84   462.9 1922.32   481.9 1929.03
#Mann= 4 ,-1 , 0
       0     .12       0   206.7     .07       0   264.3    .045       0
   292.4     .12       0
Bank Sta=264.3,292.4
XS Rating Curve= 0 ,0
Exp/Cntr=0.3,0.1

Type RM Length L Ch R = 1 ,12904.6 ,291.6,292.7,289.2
XS GIS Cut Line= 4
     1830457.164      179704.565     1830342.653      179736.144
      1830140.83      179729.633     1830004.655       179665.08
#Sta/Elev= 29
       0 1917.85     9.1 1915.79    18.3 1914.25    27.4 1913.08    45.7 1910.94
      64 1908.63    91.4 1904.93  113.861901.768     138 1898.44   147.6  1896.3
   157.2 1893.98   166.9 1892.88   176.5 1893.07   186.1 1893.54   195.7 1893.65
  202.571893.707   224.6 1894.16   243.8 1894.88   311.1 1898.26   330.1 1899.02
   367.8 1900.35   377.2  1900.9   386.6 1902.45   396.1 1905.57   405.5  1909.6
   414.9 1913.73   424.3 1917.57   433.7 1921.03   471.4 1933.92
#Mann= 5 ,-1 , 0
       0     .12       0  113.86     .07       0   157.2    .045       0
   195.7     .07       0  202.57     .12       0
Bank Sta=157.2,195.7
XS Rating Curve= 0 ,0
Exp/Cntr=0.3,0.1

Type RM Length L Ch R = 1 ,12611.9 ,266,261.3,262
XS GIS Cut Line= 3
     1830413.073      179478.071     1830176.856      179469.548
     1830086.988       179448.54
#Sta/Elev= 26
       0 1918.73    18.9 1916.45   23.981915.514    28.4  1914.7    37.8 1912.51
    75.6 1903.45    85.1 1901.28    94.6 1899.49     104 1898.23   151.3  1893.8
   160.7 1892.85   170.2    1892   179.6 1891.61   189.1 1891.77   198.6  1892.6
     208 1894.06   217.5 1896.01   226.9  1898.5   236.4 1901.61   245.6 1905.34
   273.3 1918.31   282.5 1922.33   291.8  1926.2     301 1930.13   310.2 1934.29
   328.7 1943.14
#Mann= 4 ,-1 , 0
       0    .016       0   23.98     .12       0   160.7    .045       0
   198.6     .12       0
Bank Sta=160.7,198.6
XS Rating Curve= 0 ,0
Exp/Cntr=0.3,0.1

Type RM Length L Ch R = 1 ,12350.6 ,266,269.9,255.7
XS GIS Cut Line= 3
     1830428.233      179278.088     1830289.349      179245.705
     1830140.201       179208.32
#Sta/Elev= 24
       0 1927.03    28.5 1917.43   38.211914.308    47.5 1912.02    66.6 1909.49
   68.951908.995    76.1 1907.49    85.6 1905.22   104.6 1900.44   114.1 1898.25
   123.6  1896.4   142.6 1893.12   152.2 1891.81   161.8 1890.96   171.4 1890.64
     181 1891.03   190.7 1892.62   200.3 1895.98   209.9 1901.11   219.5 1905.37
   229.1 1907.85   277.2 1918.01   286.8 1920.21   296.4 1922.83
#Mann= 5 ,-1 , 0
       0     .12       0   38.21    .016       0   68.95     .12       0
   152.2    .045       0   190.7     .12       0
Bank Sta=152.2,190.7
XS Rating Curve= 0 ,0
Exp/Cntr=0.3,0.1

Type RM Length L Ch R = 1 ,12080.7 ,267.7,264.6,256
XS GIS Cut Line= 2
     1830444.685      179037.482     1830150.422      179025.582
#Sta/Elev= 24
       0 1927.95    39.3 1915.77    49.1  1912.6    58.9 1909.91   61.441909.495
    68.7 1908.31    78.5 1907.03    88.4 1905.06   92.891904.015    98.2 1902.78
     108 1900.81   127.6  1897.4   137.4 1895.14   147.2 1892.42   157.1 1890.63
   166.9  1890.9   176.7 1894.17   186.5 1899.63   196.3  1904.5   206.2 1907.75
     216 1910.26   235.6 1915.07   284.7 1926.73   294.5 1929.26
#Mann= 5 ,-1 , 0
       0     .12       0   61.44    .016       0   92.89     .12       0
   147.2    .045       0   176.7     .12       0
Bank Sta=147.2,176.7
XS Rating Curve= 0 ,0
Exp/Cntr=0.3,0.1

Type RM Length L Ch R = 1 ,11816.1 ,239.4,229.2,222
XS GIS Cut Line= 2
      1830428.72      178788.268     1830150.422       178792.16
#Sta/Elev= 26
       0 1923.09     9.6 1919.51    19.2 1915.82    28.8 1912.27    38.4  1909.2
      48 1906.95   53.541906.217    57.6 1905.68    67.2  1904.8    76.8 1902.57
   86.691898.134      96 1893.13   105.6 1889.89   105.9 1889.86   115.2 1889.09
   124.8 1889.35   134.4 1890.27     144  1891.7   153.6 1893.26   163.2  1895.2
  169.221896.761     192 1902.99   220.7  1910.2   230.3 1912.72   249.5 1918.12
   278.3 1926.47
#Mann= 6 ,-1 , 0
       0     .12       0   53.54    .016       0   86.69     .12       0
   105.9    .045       0   134.4     .12       0  169.22     .06       0
Bank Sta=105.9,134.4
XS Rating Curve= 0 ,0
Exp/Cntr=0.3,0.1

Type RM Length L Ch R = 1 ,11587   ,181.1,194,203.4
XS GIS Cut Line= 2
     1830362.452       178541.24     1830107.867      178618.019
#Sta/Elev= 19
       0 1911.61     9.5  1909.8   26.371908.281    28.5 1908.09      38 1906.67
   46.851905.049   84.591898.086      95 1896.16   104.5 1894.16     114 1891.66
   123.5 1889.38     133 1888.53   142.4 1889.67     152 1893.46   161.4 1898.28
   170.9 1902.02   199.4 1911.56  233.341923.434   265.9 1934.81
#Mann= 7 ,-1 , 0
       0    .016       0   26.37     .12       0   46.85     .06       0
   84.59     .12       0     114    .045       0     152     .12       0
  233.34     .06       0
Bank Sta=114,152
XS Rating Curve= 0 ,0
Exp/Cntr=0.3,0.1

Type RM Length L Ch R = 1 ,11393   ,209.1,224.6,243.4
XS GIS Cut Line= 3
     1830326.947      178399.456     1830193.924      178392.805
     1830006.815      178400.758
#Sta/Elev= 20
       0 1915.41    66.6 1901.19   95.031895.264   104.6 1893.12   114.2 1890.63
   123.7 1888.54   133.2 1887.81   142.6 1889.55   151.9 1894.49   161.3 1899.96
   170.6 1903.24     180 1905.74   189.4 1908.02   198.7 1909.91  202.581910.525
   208.1  1911.4   217.5 1912.72   264.3 1919.18   301.7 1924.52   320.5  1927.3
#Mann= 5 ,-1 , 0
       0     .06       0   95.03     .12       0   114.2    .045       0
   142.6     .12       0  202.58     .06       0
Bank Sta=114.2,142.6
XS Rating Curve= 0 ,0
Exp/Cntr=0.3,0.1

Type RM Length L Ch R = 1 ,11168.4 ,138.2,111.4,84.7
XS GIS Cut Line= 2
     1830339.617      178228.446     1830061.397      178092.175
#Sta/Elev= 23
       0 1911.13    8.661909.175    38.7 1902.44    77.4 1894.12    87.1 1891.84
   106.5  1886.5   116.2 1885.13   125.9 1885.33   145.2 1887.03   164.6 1888.22
  179.941888.953   193.6 1889.66   203.3 1891.95     213 1895.65  223.621900.149
     242  1907.9   251.7 1911.84   261.4 1915.73   271.1 1919.49   280.8 1923.08
   290.4 1926.13   300.1 1928.63   309.8 1930.86
#Mann= 6 ,-1 , 0
       0    .016       0    8.66     .12       0   106.5    .045       0
   145.2     .12       0  179.94    .016       0  223.62     .12       0
Bank Sta=106.5,145.2
XS Rating Curve= 0 ,0
Exp/Cntr=0.3,0.1

Type RM Length L Ch R = 1 ,11056.9 ,74.1,65,58.9
XS GIS Cut Line= 4
      1830393.87      178144.481     1830307.716      178060.911
     1830174.252      178094.548     1830095.141      178033.687
#Sta/Elev= 30
       0 1909.56    3.481909.076    27.7 1905.78    36.9 1904.18   47.88 1902.03
   56.581900.176    64.6 1898.52    83.1 1895.23    92.3 1893.98   101.6 1892.89
   129.9 1890.12   139.7 1888.89   149.5 1887.19   159.4 1885.66   169.2 1885.29
     179  1886.1   188.8 1887.32   198.61888.419   208.5 1889.29   228.2 1890.25
     238    1891   247.8 1892.78   257.7  1895.7  263.061898.368     303 1918.22
   312.1 1922.66   321.2 1926.79   330.3 1930.08   339.3  1932.7   357.5 1937.53
#Mann= 8 ,-1 , 0
       0     .06       0    3.48    .016       0   47.88     .06       0
   56.58     .12       0   149.5    .045       0   188.8     .12       0
   198.6    .016       0  263.06     .12       0
Bank Sta=149.5,188.8
XS Rating Curve= 0 ,0
Exp/Cntr=0.3,0.1

Type RM Length L Ch R = 1 ,10992   ,12.4,62.5,108.9
XS GIS Cut Line= 4
     1830415.571       178081.31     1830328.766      177997.109
     1830195.302      178030.746     1830127.105      177978.281
#Sta/Elev= 30
       0 1903.96    18.6 1900.11   25.511898.825    37.2 1896.83    46.5 1895.62
    55.8 1894.25    65.1 1892.55    74.4 1890.69    83.7 1889.35      93 1888.61
   111.6 1888.01  120.381887.472   150.4 1886.45   160.3 1885.89   170.1  1885.5
   179.9 1885.56   189.8  1886.3   199.6 1888.22   209.4 1890.86   219.2 1892.88
   229.1 1894.67   238.9 1896.81   248.7 1899.47   258.6 1902.74   268.1 1907.58
   287.2 1917.08   296.8 1921.49   306.4 1925.18     335 1934.32   344.6 1937.49
#Mann= 5 ,-1 , 0
       0     .06       0   25.51    .016       0  120.38     .12       0
   150.4    .045       0   189.8     .12       0
Bank Sta=150.4,189.8
XS Rating Curve= 0 ,0
Exp/Cntr=0.3,0.1

Type RM Length L Ch R = 1 ,10929.5 ,9,33.6,66.7
XS GIS Cut Line= 2
     1830421.908      178075.321     1830230.936      177877.838
#Sta/Elev= 24
       0 1904.46    29.4 1898.17   33.061897.569    39.2 1896.56    58.9 1894.26
    68.7 1892.66    78.5 1890.86    88.3  1889.5    98.1 1888.75   107.9 1888.38
  114.08 1887.97   117.7 1887.73   127.6 1886.47   137.4 1885.35   147.2 1886.99
   147.9 1887.29     157 1891.25   166.8 1896.17   176.6 1900.51     206 1911.37
   225.7 1918.42   235.5 1921.85   255.1 1928.46   274.7 1935.18
#Mann= 5 ,-1 , 0
       0     .06       0   33.06    .016       0  114.08     .12       0
   117.7    .045       0   147.9     .12       0
Bank Sta=117.7,147.9
XS Rating Curve= 0 ,0
Exp/Cntr=0.3,0.1

Type RM Length L Ch R = 1 ,10895.9 ,85.2,103.8,114.5
XS GIS Cut Line= 3
     1830425.641      178067.421     1830350.988      177989.296
      1830354.46      177803.532
#Sta/Elev= 28
       0 1904.28    19.6 1899.97    29.5 1897.98    33.11897.414    39.3 1896.44
    49.1 1895.26    58.9 1894.27    68.8 1892.84    78.6 1891.19    88.4 1889.97
  106.561888.852   117.8 1888.17   127.6 1886.79   137.4 1885.63   147.2 1885.67
     157 1887.25   166.7 1890.16   176.5  1893.9   186.3 1897.46   196.1  1900.6
   205.8 1902.98   215.6  1904.5   235.2 1906.66     245 1908.05   264.5 1911.23
   274.3 1912.99   284.1  1914.9   293.8 1916.92
#Mann= 5 ,-1 , 0
       0     .06       0    33.1    .016       0  106.56     .12       0
   127.6    .045       0     157     .12       0
Bank Sta=127.6,157
XS Rating Curve= 0 ,0
Exp/Cntr=0.3,0.1

Type RM Length L Ch R = 1 ,10792.1 ,133.9,90.2,46.2
XS GIS Cut Line= 3
     1830489.147      178030.622     1830427.594      177966.206
     1830431.066      177780.442
#Sta/Elev= 28
       0 1911.91     8.9 1909.57    17.8 1907.55    53.5 1899.66   62.381897.804
   64.891897.302    71.3 1896.02    80.2 1894.58    89.1 1893.66    98.9 1893.02
   108.6 1892.19  115.571891.365   118.4 1891.03   128.2 1889.51     138 1887.76
   147.8 1886.24   157.6 1885.46   167.3 1885.34   177.1 1885.84   186.9 1886.95
   196.7  1888.7   206.4 1891.06   216.2 1893.18     226 1894.89   235.8 1896.47
  247.021898.064   255.3 1899.08   274.9  1901.1
#Mann= 7 ,-1 , 0
       0     .06       0   62.38     .12       0   64.89    .016       0
  115.57     .12       0   147.8    .045       0   177.1     .12       0
  247.02    .016       0
Bank Sta=147.8,177.1
XS Rating Curve= 0 ,0
Exp/Cntr=0.3,0.1

Type RM Length L Ch R = 1 ,10701.9 ,253.6,220.2,171.1
XS GIS Cut Line= 2
     1830577.289      177911.231     1830432.325      177763.515
#Sta/Elev= 28
       0 1911.95     9.4 1909.34    18.8 1906.63   20.481906.167    28.2 1904.04
    37.6 1901.99      47 1900.73    56.4 1899.73   65.061898.376    65.8 1898.26
    75.3 1896.33    84.7 1893.97    94.1 1891.75   103.5 1889.29   112.9 1886.93
   121.9 1885.43   122.3 1885.36   131.7 1885.22   136.9 1885.94   141.1 1886.52
   150.5 1889.41   159.9 1892.36   169.3 1894.74   178.7  1896.5   188.2 1898.37
  194.811899.819   197.6 1900.43     207 1902.42
#Mann= 6 ,-1 , 0
       0     .06       0   20.48    .016       0   65.06     .12       0
   112.9    .045       0   141.1     .12       0  194.81    .016       0
Bank Sta=112.9,141.1
XS Rating Curve= 0 ,0
Exp/Cntr=0.3,0.1

Type RM Length L Ch R = 1 ,10481.7 ,265.9,270.9,289.7
XS GIS Cut Line= 3
     1830743.366      177633.547     1830514.713      177654.381
     1830439.269      177626.558
#Sta/Elev= 27
       0 1917.64    19.1    1912   57.051901.338    76.5 1895.94    86.1 1893.65
   105.2 1889.64   114.8 1887.28   124.4 1885.44   133.9 1884.85   143.5 1885.29
   162.6 1887.12   181.8 1889.18   191.3 1890.44   210.5  1893.2     220 1894.47
   229.6 1895.92   238.5 1898.05   247.5 1900.64   256.4 1903.31   265.3 1905.78
  268.47  1906.4   274.3 1907.54   283.2  1908.8   292.1 1910.79   301.1 1913.92
  305.411915.765     310 1917.73
#Mann= 6 ,-1 , 0
       0     .06       0   57.05     .12       0   114.8    .045       0
   162.6     .12       0  268.47    .016       0  305.41     .12       0
Bank Sta=114.8,162.6
XS Rating Curve= 0 ,0
Exp/Cntr=0.3,0.1

Type RM Length L Ch R = 1 ,10210.9 ,317.6,317.9,316.2
XS GIS Cut Line= 2
     1830755.895      177399.487     1830454.832      177397.321
#Sta/Elev= 25
       0 1937.71    19.4 1930.97    29.1  1927.5    38.8 1923.86    48.6 1920.11
    77.7 1908.52    97.1 1900.98   106.8 1897.29   116.5  1894.4  123.861893.131
   126.3 1892.71     136 1891.56   145.7 1890.54   155.4  1889.4   165.1  1888.1
   174.8 1886.58   184.5 1884.98   194.2    1884     204 1884.06   213.7 1885.92
   252.5 1898.66   262.2 1901.99   281.6 1908.81  291.141912.052   301.1  1914.5
#Mann= 5 ,-1 , 0
       0     .06       0  123.86     .12       0   174.8    .045       0
   213.7     .12       0  291.14    .016       0
Bank Sta=174.8,213.7
XS Rating Curve= 0 ,0
Exp/Cntr=0.3,0.1

Type RM Length L Ch R = 1 ,9893    ,290.4,306.3,324.2
XS GIS Cut Line= 3
     1830766.448      177089.485     1830596.822      177088.124
     1830458.834      177093.297
#Sta/Elev= 23
       0  1938.8    18.8 1932.83    28.3 1929.64    37.7 1926.31    47.1 1922.82
      66 1915.51    94.2 1904.14  109.381898.233   113.1  1896.8   122.5  1893.4
   131.9  1890.4   141.4 1887.66   150.8 1885.09   160.2 1883.61   178.8 1883.75
     188 1884.35   197.2  1885.9   234.1 1892.99   252.5 1896.76   261.7 1899.04
   270.9 1901.85   280.1 1905.07   307.7  1915.3
#Mann= 4 ,-1 , 0
       0     .06       0  109.38     .12       0   150.8    .045       0
     188     .12       0
Bank Sta=150.8,188
XS Rating Curve= 0 ,0
Exp/Cntr=0.3,0.1

Type RM Length L Ch R = 1 ,9586.6  ,238.3,237.9,236.8
XS GIS Cut Line= 4
     1830809.188      176889.879     1830717.221      176839.557
     1830568.783      176771.848     1830496.946      176776.664
#Sta/Elev= 30
       0 1932.21     9.5 1929.98    19.1 1927.62    28.6 1924.96    38.1 1921.96
    57.2 1915.62    85.8  1905.7   114.4 1895.62     124 1892.43   133.6    1890
   143.2 1888.57   152.8 1887.65   181.6 1885.29   191.2 1884.38   200.8  1883.8
   210.4 1883.65     220 1884.18   223.2 1885.17   229.6 1887.14   248.8 1897.94
   258.4  1902.6     268 1906.88     277 1909.99     286 1912.82     295 1915.38
     304 1917.73     313 1919.92     322 1921.84     331 1923.54     340 1925.12
#Mann= 3 ,-1 , 0
       0     .12       0   191.2    .045       0   223.2     .12       0
Bank Sta=191.2,223.2
XS Rating Curve= 0 ,0
Exp/Cntr=0.3,0.1

Type RM Length L Ch R = 1 ,9348.8  ,333.5,312.3,291.2
XS GIS Cut Line= 4
     1830901.272      176748.957     1830790.137      176612.994
     1830670.346      176560.911     1830584.612      176570.391
#Sta/Elev= 30
       0 1934.53     9.8 1933.28    29.3 1931.24      39 1930.02    58.5 1926.66
    68.3 1924.32      78 1921.52    87.8 1918.22   117.1 1907.61   126.8 1904.25
   136.6 1901.17   146.3 1898.69   156.1 1896.76   184.9 1891.91   194.3    1890
   203.6 1887.51   212.9  1884.8   222.3 1883.72   231.6 1883.64   240.9 1884.69
   250.2 1887.09   259.6 1889.74   287.6 1896.76   296.9 1899.42   325.4 1908.55
   344.6 1915.08   363.7 1922.64   373.3 1926.28   382.9  1929.4   392.5 1932.02
#Mann= 3 ,-1 , 0
       0     .12       0   212.9    .045       0   240.9     .12       0
Bank Sta=212.9,240.9
XS Rating Curve= 0 ,0
Exp/Cntr=0.3,0.1

Type RM Length L Ch R = 1 ,9036.5  ,240.6,247.9,254.9
XS GIS Cut Line= 3
     1831002.383       176297.88     1830732.846      176336.953
     1830614.819      176379.557
#Sta/Elev= 30
       0 1934.27     9.7 1930.59    19.4 1926.57    29.2    1923    58.4 1912.93
    68.1 1909.51     107  1895.4   116.7 1891.54   126.4 1887.35   135.8  1884.6
   136.2 1884.48   145.9 1883.55   155.6 1883.48   165.4 1883.61   175.1 1883.85
   184.8 1884.23   204.3 1885.21     214 1885.87   223.7 1887.91   233.4 1891.83
   243.2 1896.25   252.9 1899.88   272.4 1905.69     282 1908.68   291.7 1911.44
   320.6 1917.43   339.9 1920.94   349.6 1922.83   368.9 1926.39   397.8 1931.88
#Mann= 3 ,-1 , 0
       0     .12       0   135.8    .045       0   165.4     .12       0
Bank Sta=135.8,165.4
XS Rating Curve= 0 ,0
Exp/Cntr=0.3,0.1

Type RM Length L Ch R = 1 ,8788.6  ,205.9,222.8,239.9
XS GIS Cut Line= 4
     1831014.004      176085.584     1830883.887      176073.932
     1830769.304      176068.723     1830702.115      176020.969
#Sta/Elev= 25
       0 1928.54    18.7    1923    37.3 1917.69    65.3 1910.18    74.6 1907.77
   102.6 1900.82   121.3 1896.36   140.2 1892.01   149.8 1889.63   159.3 1886.62
   168.9 1884.24   178.4 1883.56     188 1884.48   197.6 1887.19   207.1  1890.1
   216.7 1892.27   235.8 1896.23   245.3 1898.57   254.5 1901.36   263.7 1904.45
     282 1911.01   300.3 1917.83   309.4 1921.31   318.6 1924.36   327.8 1926.82
#Mann= 3 ,-1 , 0
       0     .12       0   159.3    .045       0   197.6     .12       0
Bank Sta=159.3,197.6
XS Rating Curve= 0 ,0
Exp/Cntr=0.3,0.1

Type RM Length L Ch R = 1 ,8565.8  ,195.8,197.9,200.1
XS GIS Cut Line= 3
     1831053.283       175955.18     1830905.906      175871.597
     1830809.016      175819.241
#Sta/Elev= 23
       0 1918.39     9.4 1915.58    18.8 1912.89    28.2 1910.32    47.1 1905.37
    56.5 1902.95    65.9 1900.79    75.3 1898.91     113 1892.08   122.4 1890.52
   131.8 1889.24     160  1886.2   169.4 1884.96   178.6 1883.92   187.8  1883.5
     197 1883.49   206.1 1884.06   215.3 1886.67   224.5 1889.81   233.7 1892.78
   242.8 1896.23     252 1900.24   279.6  1913.8
#Mann= 3 ,-1 , 0
       0     .12       0   178.6    .045       0   206.1     .12       0
Bank Sta=178.6,206.1
XS Rating Curve= 0 ,0
Exp/Cntr=0.3,0.1

Type RM Length L Ch R = 1 ,8367.9  ,279.5,264.4,249.8
XS GIS Cut Line= 2
     1831123.165       175775.51     1830906.151      175640.962
#Sta/Elev= 29
       0 1911.56     9.8 1909.22    19.6 1906.89    29.5 1904.59    39.3 1902.33
    49.1 1900.06    58.9 1897.85    68.8 1895.93    78.6 1894.34    88.4 1893.06
    98.2  1891.9     108 1890.75   117.8 1889.61   127.7 1888.04   137.5  1885.9
   147.3 1884.14   149.8 1884.01   157.1 1883.62   164.8 1884.62     167  1884.9
   176.8 1888.61   186.6 1893.12   196.4 1897.07   206.2 1901.08   216.1 1905.22
   225.9 1909.38   235.7 1913.53   245.5 1917.73   255.3 1921.87
#Mann= 3 ,-1 , 0
       0     .12       0   137.5    .045       0     167     .12       0
Bank Sta=137.5,167
XS Rating Curve= 0 ,0
Exp/Cntr=0.3,0.1

Type RM Length L Ch R = 1 ,8103.5  ,307.1,299.6,291.6
XS GIS Cut Line= 3
     1831281.094      175501.226       1831130.7       175475.77
     1830986.648       175445.03
#Sta/Elev= 29
       0 1916.69     9.5 1914.84    38.1 1909.58    47.7  1907.7    57.2 1905.69
    66.7 1903.54    76.3 1901.22    85.8 1898.73    95.3 1896.05   104.9 1893.15
   114.4 1889.62   123.9 1885.67   131.8 1883.89   133.5 1883.51     143 1883.45
   152.5 1883.64   162.4 1884.56     182 1887.54   191.8 1889.26   201.6 1891.18
   211.4 1893.41   221.3 1895.93   231.1 1898.75   240.9 1901.89   250.7 1905.35
   260.6 1909.15   270.4 1913.21     290 1921.58   299.8  1925.6
#Mann= 3 ,-1 , 0
       0     .12       0   131.8    .045       0   162.4     .12       0
Bank Sta=131.8,162.4
XS Rating Curve= 0 ,0
Exp/Cntr=0.3,0.1

Type RM Length L Ch R = 1 ,7803.9  ,354.4,348.7,342.6
XS GIS Cut Line= 3
     1831314.296       175178.34     1831037.533      175188.515
     1831003.752      175190.518
#Sta/Elev= 24
       0 1925.95    19.1 1920.82    28.6    1918    38.2 1914.87    47.8 1911.58
    76.4 1901.58      86 1898.32    95.5  1895.4     105  1893.3   114.6 1891.86
   133.7 1889.55   152.8 1887.42   181.4  1884.5     191 1883.76   200.6 1883.49
   210.1 1883.46   229.2 1883.45   238.8 1883.95   248.3 1885.94   267.4 1892.18
     277 1895.24   285.4 1898.05   293.9 1901.09   310.8 1907.54
#Mann= 3 ,-1 , 0
       0     .12       0   210.1    .045       0   238.8     .12       0
Bank Sta=210.1,238.8
XS Rating Curve= 0 ,0
Exp/Cntr=0.3,0.1

Type RM Length L Ch R = 1 ,7455.2  ,280.9,280,278.4
XS GIS Cut Line= 2
     1831329.827      174869.821     1830997.466      174931.772
#Sta/Elev= 29
       0 1924.66     9.7  1922.1      29 1916.84    48.3 1911.44    86.9 1900.43
   106.3 1895.04   115.9 1891.67   125.6 1887.45   135.2 1883.65   137.7  1883.2
   144.9  1881.9   154.6 1881.96   164.2 1882.54   173.9 1883.02   183.5 1883.24
   212.5 1883.56   222.2 1883.78   231.8 1884.18   241.5 1884.78   251.2 1885.64
   260.8 1886.75   270.5 1888.07   280.1 1889.58   289.8 1891.33   299.4 1893.34
   309.1  1895.6   318.8  1898.1   328.4 1900.82   338.1 1903.68
#Mann= 3 ,-1 , 0
       0     .12       0   137.7    .045       0   164.2     .12       0
Bank Sta=137.7,164.2
XS Rating Curve= 0 ,0
Exp/Cntr=0.3,0.1

Type RM Length L Ch R = 1 ,7175.1  ,361.2,370.4,381.5
XS GIS Cut Line= 3
       1831336.7      174605.954     1831215.558      174610.307
     1830973.201      174664.164
#Sta/Elev= 27
       0 1937.09     9.3 1933.53    18.6 1929.73      28 1925.67    46.6 1917.44
    93.2 1897.14   102.6 1893.15   111.9 1889.89   121.2 1887.89   149.9  1884.3
   159.4 1882.91     169 1881.23   178.5 1879.71   188.1 1879.22   197.6  1880.2
   207.2 1881.89   216.7 1883.42   226.3 1884.58   235.8 1885.62   264.4 1888.42
   283.6 1890.42   293.1 1891.54   312.2    1894   331.3 1896.79   340.8 1898.31
   350.4 1899.98   369.5  1903.6
#Mann= 3 ,-1 , 0
       0     .12       0     169    .045       0   197.6     .12       0
Bank Sta=169,197.6
XS Rating Curve= 0 ,0
Exp/Cntr=0.3,0.1

Type RM Length L Ch R = 1 ,6804.8  ,205.2,206.4,202.5
XS GIS Cut Line= 3
     1831316.418      174291.175     1831095.203      174296.799
     1830960.138      174280.112
#Sta/Elev= 26
       0 1910.34     9.6 1906.74    19.2 1903.26    28.9 1900.04    38.5  1897.1
    48.1 1894.37    57.7 1891.93    67.4 1889.79      77 1887.88    86.6 1886.12
    96.2 1884.46   105.8 1882.54   125.1 1878.02   134.7 1876.92   144.3  1877.2
   153.9 1877.96   163.6 1878.57   173.2 1878.96     202 1879.91   260.2 1882.31
   269.9 1883.25   279.6 1885.39   289.3 1888.55     299 1892.01   318.5  1898.8
   357.4 1912.08
#Mann= 3 ,-1 , 0
       0     .12       0   125.1    .045       0   153.9     .12       0
Bank Sta=125.1,153.9
XS Rating Curve= 0 ,0
Exp/Cntr=0.3,0.1

Type RM Length L Ch R = 1 ,6598.3  ,269.4,286.9,306.3
XS GIS Cut Line= 4
      1831314.55      174199.712     1831124.717      174137.077
     1831011.842      174138.863      1830973.58      174129.539
#Sta/Elev= 25
       0 1902.01     9.5 1899.45      19  1897.4    28.6  1895.8    76.2 1889.64
    95.2 1887.47   104.7 1886.54   114.2 1885.73   152.3 1882.76   171.3 1881.37
   199.9 1879.46   237.5 1877.62   246.9 1876.99   256.3 1876.01   265.8 1874.77
   275.2 1874.11   284.6 1875.85     294 1880.16   303.4 1884.65   312.8 1888.24
   320.7 1890.76   328.5 1893.57   336.4 1896.66   344.3 1900.02   352.2 1903.61
#Mann= 3 ,-1 , 0
       0     .12       0   256.3    .045       0   284.6     .12       0
Bank Sta=256.3,284.6
XS Rating Curve= 0 ,0
Exp/Cntr=0.3,0.1

Type RM Length L Ch R = 1 ,6311.5  ,213.6,214.1,214.7
XS GIS Cut Line= 3
     1831391.933      174028.687     1831260.134      173966.938
      1831094.01      173873.734
#Sta/Elev= 20
       0 1903.14    19.4 1898.77    58.2 1890.34    77.6  1885.9      97  1881.3
   106.7 1879.14   116.4  1877.5   126.1 1876.36   155.1 1873.42   193.2 1869.99
   202.7 1869.29   212.2 1869.09   221.7 1869.96   231.3 1872.07   259.8 1880.31
   278.9 1885.68   297.9 1890.47     317  1894.9   326.5 1897.28     336 1899.91
#Mann= 3 ,-1 , 0
       0     .12       0   193.2    .045       0   221.7     .12       0
Bank Sta=193.2,221.7
XS Rating Curve= 0 ,0
Exp/Cntr=0.3,0.1

Type RM Length L Ch R = 1 ,6097.4  ,317.7,314.6,311.4
XS GIS Cut Line= 3
     1831486.484      173853.721      1831336.87      173768.858
     1831213.644      173698.641
#Sta/Elev= 24
       0 1903.51    19.1 1899.48    38.2 1895.28    66.9 1888.72      86 1884.25
    95.6 1882.12   105.1 1880.23   143.3 1873.74   152.9 1871.88   162.4 1869.61
     172 1867.26   181.5 1866.73   190.9 1868.17   200.4 1870.09   209.8 1871.68
   219.3 1872.87   238.2 1874.74   247.6 1875.85   257.1 1877.09   266.6 1878.48
   285.5 1881.55   294.9 1883.18   304.4 1884.98   313.8 1886.99
#Mann= 3 ,-1 , 0
       0     .12       0   162.4    .045       0   200.4     .12       0
Bank Sta=162.4,200.4
XS Rating Curve= 0 ,0
Exp/Cntr=0.3,0.1

Type RM Length L Ch R = 1 ,5782.8  ,295.3,275.8,256.4
XS GIS Cut Line= 3
     1831646.467      173612.324     1831553.536       173532.91
     1831377.371      173446.638
#Sta/Elev= 26
       0 1898.11    18.8 1893.36    28.2 1890.81    56.4 1882.68    65.8 1880.05
    84.6 1875.36      94 1872.71   103.4 1869.88   112.8 1867.78     132  1865.6
   141.9 1864.07   151.7 1862.75   161.5 1862.18   171.3 1862.07   181.1 1862.21
   190.9 1862.69   220.3 1864.97   230.1 1865.87   239.9    1867   249.7 1868.38
   259.6 1869.94   269.4 1871.64     289 1875.29   298.8 1877.19   308.6 1879.31
   318.4  1881.6
#Mann= 3 ,-1 , 0
       0     .12       0   151.7    .045       0   190.9     .12       0
Bank Sta=151.7,190.9
XS Rating Curve= 0 ,0
Exp/Cntr=0.3,0.1

Type RM Length L Ch R = 1 ,5507    ,180.8,186.9,193
XS GIS Cut Line= 3
     1831738.218      173301.894     1831685.698      173263.379
     1831400.422      173284.941
#Sta/Elev= 29
       0 1882.19     9.3 1879.45    18.6 1876.84    27.9 1874.41    37.2 1872.33
    46.5 1870.56    65.1 1867.36    84.2 1864.72    93.7 1863.22   112.8 1859.57
   117.8 1858.98   122.4 1858.44   131.9 1858.22     151 1858.31     170 1858.16
   198.6  1857.8   217.7 1857.87   227.2 1858.09   236.8 1858.48   246.3 1859.04
   255.9 1859.82   265.4 1860.82   274.9 1862.07   284.5 1864.25     294 1867.27
   313.1 1873.76   332.2 1880.81   341.7 1884.16   351.2 1887.33
#Mann= 3 ,-1 , 0
       0     .12       0   117.8    .045       0     151     .12       0
Bank Sta=117.8,151
XS Rating Curve= 0 ,0
Exp/Cntr=0.3,0.1

Type RM Length L Ch R = 1 ,5320.1  ,185.4,199.8,215.4
XS GIS Cut Line= 3
     1831767.794      173138.411     1831697.851      173087.598
     1831418.042      173065.213
#Sta/Elev= 21
       0 1873.37     9.6 1872.78    19.2 1872.08    38.4 1870.16      48  1868.9
    57.6 1867.55    67.2 1865.73    86.4  1862.3   125.2 1856.55   134.8 1855.26
   144.5 1854.51   154.2 1854.34   173.6 1854.58   192.9 1854.71   260.7  1854.8
   309.1 1855.07   318.8 1854.92   328.4 1856.43   338.1 1861.33   347.8 1868.35
   367.2 1883.36
#Mann= 3 ,-1 , 0
       0     .12       0   134.8    .045       0   173.6     .12       0
Bank Sta=134.8,173.6
XS Rating Curve= 0 ,0
Exp/Cntr=0.3,0.1

Type RM Length L Ch R = 1 ,5120.2  ,372.3,375.7,360.8
XS GIS Cut Line= 4
      1831808.26       172954.82     1831693.608      172926.856
     1831516.525      172856.543     1831472.841      172856.543
#Sta/Elev= 24
       0 1872.66     9.8 1870.46    19.7 1868.72    49.2 1864.62    98.3 1858.41
     118 1856.22   127.5 1855.08   146.6  1853.1   156.1 1852.22   165.6 1851.44
   175.2 1850.78   184.7 1850.25   203.8  1849.4   222.8 1848.35   232.3 1848.53
   241.9 1849.28   260.9 1851.35     280 1853.02   289.5 1854.35     299 1856.45
   308.5 1859.44   317.3 1862.32   334.8 1868.71   352.2 1875.17
#Mann= 3 ,-1 , 0
       0     .12       0   203.8    .045       0   241.9     .12       0
Bank Sta=203.8,241.9
XS Rating Curve= 0 ,0
Exp/Cntr=0.3,0.1

Type RM Length L Ch R = 1 ,4744.5  ,372.6,330.4,304.8
XS GIS Cut Line= 4
     1831937.252      172712.192      1831844.65      172684.668
       1831688.4      172583.106     1831580.071       172587.92
#Sta/Elev= 24
       0 1878.35     9.7 1874.77    19.3 1871.54    38.6 1865.64    48.3 1862.46
      58 1859.06    67.6 1856.16    77.3 1854.37    96.6 1852.36   145.6  1846.2
   155.5 1845.14   165.3 1845.13   175.1 1845.89   184.9 1847.04   194.7 1848.08
   204.5 1848.87   214.3 1849.44   224.1 1849.81   243.7 1850.18     292 1850.45
     301 1850.81   310.1 1851.61   328.1 1853.85   391.4 1861.47
#Mann= 3 ,-1 , 0
       0     .12       0   145.6    .045       0   175.1     .12       0
Bank Sta=145.6,175.1
XS Rating Curve= 0 ,0
Exp/Cntr=0.3,0.1

Type RM Length L Ch R = 1 ,4414.2  ,266.5,281.8,296.9
XS GIS Cut Line= 4
     1832006.905      172286.608      1831930.49      172294.629
     1831741.253       172405.74     1831601.491       172416.44
#Sta/Elev= 30
       0 1885.47    19.2 1876.55    38.4 1867.34    57.6 1858.04    67.2 1853.28
    76.8 1848.33    86.4 1844.12    95.9 1841.99   105.5 1842.08     115 1842.77
   124.5 1843.12   143.6  1843.3   153.2 1843.24   162.7 1842.91   172.2 1841.88
   181.8 1840.64   191.3 1841.74   200.9 1843.24   210.4 1844.01     220 1844.39
     239 1844.71   286.7 1844.98   333.7 1845.05   352.4 1845.25   361.7 1845.48
   380.4  1846.3   389.7 1846.92   417.8 1849.27   427.1 1850.15   436.4  1851.2
#Mann= 3 ,-1 , 0
       0     .12       0   162.7    .045       0   200.9     .12       0
Bank Sta=162.7,200.9
XS Rating Curve= 0 ,0
Exp/Cntr=0.3,0.1

Type RM Length L Ch R = 1 ,4132.4  ,291.7,289.6,287.4
XS GIS Cut Line= 3
     1831988.315      172095.765     1831896.733      172080.501
     1831583.285      172120.422
#Sta/Elev= 16
       0 1881.98    18.6  1874.9    74.3 1852.91    92.8  1845.8   102.4 1842.18
     112 1839.19   121.6 1837.69   131.2 1837.39   207.8 1836.97   265.2  1836.5
   284.4 1836.23   293.9 1836.61   303.5 1837.53   313.1 1838.59   322.6 1839.52
   408.8 1847.31
#Mann= 3 ,-1 , 0
       0     .12       0   265.2    .045       0   293.9     .12       0
Bank Sta=265.2,293.9
XS Rating Curve= 0 ,0
Exp/Cntr=0.3,0.1

Type RM Length L Ch R = 1 ,3842.8  ,222.6,207.9,194.2
XS GIS Cut Line= 3
     1831932.975       171786.71      1831845.42      171825.879
      1831541.02      171866.713
#Sta/Elev= 30
       0 1868.39     9.6 1865.76    19.2 1862.91    38.4  1856.9    57.6  1850.7
    76.7 1844.78    86.3 1842.03    95.9 1839.52   105.5  1837.3   115.1 1835.44
   124.7  1833.9   143.9 1831.27   153.5 1830.31   163.1 1830.01   172.7  1830.6
   182.3 1831.53   191.9  1832.2   201.5 1832.55   230.3 1832.87   239.9  1832.8
   268.7 1832.26   278.3 1832.27   287.9 1832.55   297.5 1833.05   326.3 1835.01
   345.5  1836.7   355.1 1837.67   374.2 1839.96   383.8 1841.27     403 1844.22
#Mann= 3 ,-1 , 0
       0     .12       0   143.9    .045       0   172.7     .12       0
Bank Sta=143.9,172.7
XS Rating Curve= 0 ,0
Exp/Cntr=0.3,0.1

Type RM Length L Ch R = 1 ,3634.9  ,246.5,253.7,259.8
XS GIS Cut Line= 3
     1831832.196      171593.213     1831661.392      171700.879
     1831519.547      171729.125
#Sta/Elev= 24
       0 1858.62    28.8 1853.03    38.5 1850.92    48.1 1847.97    57.7 1844.67
    67.3 1841.19    76.9 1837.49    86.5 1833.42    96.2 1829.14   105.6 1826.16
   115.4 1825.27     125 1825.53   134.6 1826.32   144.2 1827.16   163.4 1828.35
   182.7 1829.25   221.2 1830.72   240.5 1831.66   269.4 1833.34     279 1834.09
   288.7 1835.48   298.3  1837.5   317.6 1842.21   346.5 1849.66
#Mann= 3 ,-1 , 0
       0     .12       0   105.6    .045       0   134.6     .12       0
Bank Sta=105.6,134.6
XS Rating Curve= 0 ,0
Exp/Cntr=0.3,0.1

Type RM Length L Ch R = 1 ,3381.2  ,115.8,147.1,178.2
XS GIS Cut Line= 2
     1831746.607      171397.087     1831467.681      171504.494
#Sta/Elev= 26
       0 1844.66    19.3 1842.72    28.9 1841.68    38.6 1840.33    48.2 1838.77
    67.5 1835.38   106.1 1828.91   115.7 1827.23   125.3 1825.42     135 1823.35
   144.6 1821.52   154.3 1820.74   163.9 1820.96   173.6 1821.58   183.2 1822.11
   192.8 1822.35   212.1 1822.58   221.8 1822.95   231.4 1823.63     241 1824.91
   250.7 1826.64   260.3 1828.91     270 1832.49   279.6 1837.52   289.2 1842.94
   298.9 1847.52
#Mann= 3 ,-1 , 0
       0     .12       0   144.6    .045       0   173.6     .12       0
#XS Ineff= 2 , 0
                          228.26         1844.97
Permanent Ineff=
       F       F
Bank Sta=144.6,173.6
XS Rating Curve= 0 ,0
Exp/Cntr=0.3,0.1

Type RM Length L Ch R = 1 ,3234.1  ,119.9,120.2,125.2
XS GIS Cut Line= 4
     1831718.925      171316.679     1831625.802      171337.598
     1831438.302      171271.626     1831387.385      171303.146
#Sta/Elev= 26
       0 1839.03     9.5  1837.9    28.6 1835.38   35.271834.574    47.7 1833.08
    76.4 1829.12    85.9 1827.92    95.4 1826.86   133.3 1823.56   152.2 1821.76
   161.7    1821   171.2 1820.85   180.6 1821.36   218.5 1825.08     228 1826.09
   237.4 1827.21   246.9 1828.49   256.4 1829.92   265.8 1831.48   275.3  1833.2
   284.8 1835.07   294.2 1837.19   319.9 1847.38     337 1853.88   345.5 1856.94
   354.1 1859.61
#Mann= 4 ,-1 , 0
       0    .016       0   35.27     .12       0   152.2    .045       0
   180.6     .12       0
Bank Sta=152.2,180.6
XS Rating Curve= 0 ,0
Exp/Cntr=0.3,0.1

Type RM Length L Ch R = 1 ,3113.9  ,167.2,132.8,94.1
XS GIS Cut Line= 4
     1831677.784      171219.263     1831612.781      171233.865
     1831425.281      171167.893     1831344.168      171218.106
#Sta/Elev= 30
       0 1843.56     9.5 1839.97      19 1836.63    28.6 1833.71    38.1 1831.17
    47.6 1828.99    57.1 1827.23    66.6 1826.03    85.6 1824.63   104.5 1823.33
   142.3 1821.26   151.8 1820.54   161.3 1819.56   170.7 1819.04   189.7 1819.32
   199.1 1819.63  221.311820.727   246.5 1821.75   255.9 1822.42   265.4  1823.3
   274.9 1825.98  279.851827.486   284.5  1828.9     294 1832.07   303.6 1835.48
   313.1  1839.1   332.2 1846.67   341.7 1850.36   351.2 1853.86   360.8 1857.08
#Mann= 5 ,-1 , 0
       0     .12       0   161.3    .045       0   189.7     .12       0
  221.31    .016       0  279.85     .12       0
Bank Sta=161.3,189.7
XS Rating Curve= 0 ,0
Exp/Cntr=0.3,0.1
